HEC-RAS study STONYCK.prj: STONYCK

--- STONYCK.g01 (geometry) --- (continued)

Type RM Length L Ch R = 1 ,22192   ,435.4,439,441.6
XS GIS Cut Line= 3
2218384.93891814464273.1015333142218588.77417943463919.003098643
2218448.96409637 463690.34174784
#Sta/Elev= 30
       0  2485.7    78.4 2487.63    92.2 2486.54   102.7 2489.76   106.1 2489.42
   115.3 2485.83     140 2482.87   161.4 2481.63   207.4 2480.74   253.8 2482.03
   401.5 2477.68   480.2  2476.8   488.9 2475.55   499.8 2472.06   509.2    2472
   513.9 2471.03   527.9 2469.77   538.4 2469.87   544.2 2470.88   556.1 2475.33
   569.1 2484.15     582 2491.27   602.9 2507.96   609.1 2514.14   622.7 2531.22
   631.1 2546.64   632.1 2547.77   649.8 2558.69   663.9 2564.41   676.6 2568.42
#Mann= 7 ,-1,0
       0     .05       0     140     .06       0     340     .05       0
  448.58     .07       0  478.58      .1       0   513.9    .045       0
   544.2      .1       0
Bank Sta=513.9,544.2
XS Rating Curve= 0 ,0
Exp/Cntr(USF)=0,0
Exp/Cntr=0.3,0.1

Type RM Length L Ch R = 1 ,21753   ,365.6,370.4,373.8
XS GIS Cut Line= 3
2218694.61171894464107.1587244462218949.40579555463729.540836549
2218820.04880281 463425.09458091
#Sta/Elev= 30
       0 2477.71   118.2 2475.84   171.3 2473.27   212.9 2473.28   231.6 2472.49
     263    2469   306.4 2469.79   328.1 2468.25   353.2 2468.72   398.1 2466.01
   436.7 2465.94     482    2462   503.7 2461.71   547.2 2463.92     595 2463.77
   612.4 2460.97   620.2 2457.74   630.6 2456.49   642.8 2456.81  646.012457.746
   660.2 2462.58     695 2463.12   712.4 2464.36   716.7 2465.03   728.2 2469.45
   746.5 2477.96   755.7 2483.68   764.5 2491.03   777.5 2505.06   786.3 2513.07
#Mann= 6 ,-1,0
       0     .06       0      30     .07       0     100     .05       0
     270      .1       0   620.2    .045       0  646.01      .1       0
#XS Ineff= 2 , 0
          561.46 2466.28
Permanent Ineff=
       F       F
Bank Sta=620.2,646.01
XS Rating Curve= 0 ,0
Exp/Cntr(USF)=0,0
Exp/Cntr=0.3,0.1

Type RM Length L Ch R = 1 ,21383   ,419.7,415.7,411.9
XS GIS Cut Line= 4
2219146.10640599463735.611756831 2219246.9231702463558.934598728
2219197.70303905463282.0671521562219095.13657864463227.318100572
#Sta/Elev= 30
       0 2460.36    36.5 2459.56   127.1 2455.76   173.4 2455.69   205.2 2454.09
   231.4 2453.91   237.7 2453.48     254 2450.78   262.5 2450.67   274.3 2451.81
282.38422449.227   293.5 2448.43305.58422449.225   314.9 2451.27     323 2451.88
   335.2 2451.46   352.2 2449.32   355.5 2449.31   363.6 2451.56   371.8 2452.13
   392.1 2450.16   424.6 2450.47   436.8 2451.92     453 2451.54   469.3 2454.68
   495.4 2453.27   522.6 2453.01   554.4 2456.09   586.1 2461.79   600.9 2466.12
#Mann= 3 ,-1,0
       0      .1       0282.3842    .045       0305.5842      .1       0
#XS Ineff= 2 , 0
                             480         2456.03
Permanent Ineff=
       F       F
Bank Sta=282.3842,305.5842
XS Rating Curve= 0 ,0
Exp/Cntr(USF)=0,0
Exp/Cntr=0.3,0.1

Type RM Length L Ch R = 1 ,20967   ,324.2,330.1,333.1
XS GIS Cut Line= 3
2219593.49562212463590.008951499 2219649.2326304463423.105416109
2219543.67512019463194.978109272
#Sta/Elev= 30
       0  2448.6      47 2444.95    68.3 2444.93    85.2  2442.8   100.8 2442.04
   144.3 2442.73   156.9 2443.98   173.8 2444.78   182.5 2444.71   187.3 2444.32
   200.1 2441.78   226.6 2439.31   241.5 2440.63   257.4 2439.84   266.2 2439.89
   279.5  2438.9   295.7 2440.04   301.8 2440.04322.17382436.013   331.9 2435.22
   341.2  2435.4344.97372435.919   358.8 2438.24   367.6 2445.16   377.1 2451.77
   394.1 2464.48   402.9 2471.21   411.7 2479.42   420.5 2486.99   427.3 2497.49
#Mann= 3 ,-1,0
       0      .1       0322.1738    .045       0344.9737      .1       0
Bank Sta=322.1738,344.9737
XS Rating Curve= 0 ,0
Exp/Cntr(USF)=0,0
Exp/Cntr=0.3,0.1

Type RM Length L Ch R = 1 ,20637   ,126.8,140.1,148.4
BEGIN DESCRIPTION:
structure xs 4
END DESCRIPTION:
XS GIS Cut Line= 3
2219724.88742353463406.1002903272219892.90385469463218.452430899
2219873.39996126463082.626320433
#Sta/Elev= 30
       0 2438.56      12 2438.16    22.8 2437.37    49.6 2437.77    82.3 2436.65
    96.5 2436.46     114 2434.79   124.7 2434.25   156.9 2434.65   164.4 2434.46
   172.9 2433.78   187.1 2434.16   199.9 2434.05   220.8 2432.74   242.8 2432.95
   289.5 2432.33   297.6 2431.41   309.7 2428.86   313.7 2428.04   317.8 2427.72
   321.9  2427.8   329.9 2428.86     338 2428.87   346.1 2429.34   349.1 2429.81
   354.2  2432.6   362.3 2436.39   380.9 2447.47   384.6 2449.12   389.1 2450.61
#Mann= 7 ,-1,0
       0      .1       0      20     .06       0     150      .1       0
     170     .05       0  271.88      .1       0   309.7    .045       0
   329.9      .1       0
Bank Sta=309.7,329.9
XS Rating Curve= 0 ,0
Exp/Cntr(USF)=0,0
Exp/Cntr=0.5,0.3

Type RM Length L Ch R = 1 ,20497   ,53.1,52.7,53.6
BEGIN DESCRIPTION:
structure xs 3; 16.3 ft between structure and xs
END DESCRIPTION:
XS GIS Cut Line= 5
2219776.87560831463405.786203299  2219805.394491463333.441069249
2219867.79627168463271.0392885722219973.66895575 463200.92492826
2220184.16619525 462846.28368375
#Sta/Elev= 30
       0 2436.54    60.8 2436.04    77.8 2435.63    96.9 2433.91   123.4 2434.35
   205.1 2431.93     293 2430.67   306.7 2428.44     316 2429.64   329.7 2430.15
   352.8 2428.84   358.9 2427.33   368.6 2423.24   371.8 2422.25   381.1 2421.84
   385.7 2421.91   390.72423.255   404.3 2431.53     409 2435.27   413.6 2437.67
   422.9 2439.43   455.2 2439.66   492.7 2441.38     502 2441.11   517.3 2442.09
   540.8  2442.2   586.5 2445.26   618.3 2446.26   660.2 2446.89   705.4 2444.89
#Mann= 6 ,-1,0
       0      .1       0      10     .06       0  117.76     .05       0
     293      .1       0   368.6    .045       0   390.7      .1       0
#XS Ineff= 4 ,-1
       0   223.1  2424.5   223.1  332.17 2430.64  332.17     352  2424.5
     407   705.4  2424.5
Permanent Ineff=
       F       F       F       F
Bank Sta=368.6,390.7
XS Rating Curve= 0 ,0
Exp/Cntr(USF)=0,0
Exp/Cntr=0.5,0.3

Type RM Length L Ch R = 1 ,20444   ,49.2,47.5,46.1
BEGIN DESCRIPTION:
structure xs 2; 23.6 ft between structure and xs
END DESCRIPTION:
XS GIS Cut Line= 5
2219805.29283414463389.6290560842219855.87683043463317.314766377
2219928.09462155463259.8209909222220035.36959282463200.223784657
  2220195.054831462927.585497369
#Sta/Elev= 30
       0 2435.66    78.7  2433.1   119.3 2432.64   139.8 2433.12     154 2432.45
   170.4 2431.21   208.1 2431.12   217.3 2430.62   244.3 2429.97   268.4 2429.77
   290.5 2430.06   303.3 2428.97     330 2427.44     347 2425.02   352.4    2423
   357.8 2421.92   360.3 2421.89   376.3  2422.4     381 2423.01   390.2 2426.74
   399.8 2429.39   422.7 2432.67   431.5 2433.61   469.1 2436.46   486.9 2439.14
   510.6 2442.08   552.5 2445.33   580.9 2446.99   598.8 2447.74   619.2  2447.7
#Mann= 5 ,-1,0
       0     .06       0      50     .05       0  300.56      .1       0
   352.4    .045       0     381      .1       0
#XS Ineff= 2 , 0
             344  2424.5     389          2424.5
Permanent Ineff=
       F       F
Bank Sta=352.4,381
XS Rating Curve= 0 ,0
Exp/Cntr(USF)=0,0
Exp/Cntr=0.5,0.3

Type RM Length L Ch R = 1 ,20397   ,95,90.8,86.4
BEGIN DESCRIPTION:
structure xs 1
END DESCRIPTION:
XS GIS Cut Line= 3
 2219857.0686819463379.4552936422220092.16222468463202.327215467
2220203.77663424462976.918333337
#Sta/Elev= 30
       0 2434.25    26.7 2433.55      49 2432.12      64 2431.78    83.5 2432.28
    92.4 2432.05   103.8 2430.54   149.5 2429.45   163.3 2428.73   176.6 2429.11
   223.8 2428.74   239.3 2430.06   255.2 2427.96   313.5 2426.97     318 2425.79
   322.4  2422.8   326.42421.767     343 2421.29   350.42421.759     367    2425
   375.5 2426.22   380.4 2428.19   384.8 2429.23   396.7 2429.65   405.7  2431.6
   425.1 2434.09   460.8 2439.92   507.2 2445.62   536.7 2447.95   545.9 2448.18
#Mann= 7 ,-1,0
       0     .05       0     220     .06       0  304.35      .1       0
   326.4    .045       0   350.4      .1       0  374.35     .05       0
  404.35      .1       0
#XS Ineff= 2 , 0
          305.58 2430.05
Permanent Ineff=
       F       F
Bank Sta=326.4,350.4
XS Rating Curve= 0 ,0
Exp/Cntr(USF)=0,0
Exp/Cntr=0.3,0.1

Type RM Length L Ch R = 1 ,20306   ,36.2,35.6,36
BEGIN DESCRIPTION:
structure xs 4
END DESCRIPTION:
XS GIS Cut Line= 3
2220049.29302564463502.9439710862220179.50911831463268.657170052
2220235.13590521462984.758151079
#Sta/Elev= 30
       0 2429.58    24.9 2428.46    35.8 2429.12    84.4 2426.85   109.3  2426.7
   154.1 2425.77   180.5 2424.34   203.2  2424.8   212.5  2425.8   221.7 2425.34
   235.4  2426.3   253.4 2425.82   261.2 2426.06     292 2425.91   300.1 2426.46
   304.2 2426.44   312.3 2425.48   316.4 2424.68   324.6  2420.2   329.5 2419.49
   339.7 2419.25   346.6 2420.17     350  2420.6   361.3 2420.83   397.7 2424.28
   410.2 2428.39   421.5 2430.49   487.6 2440.65   524.3 2447.04   557.3 2450.31
#Mann= 6 ,-1,0
       0     .05       0     120      .1       0     170     .05       0
   324.6    .045       0   346.6     .05       0  438.04      .1       0
#XS Ineff= 1 ,-1
   68.62  244.39 2426.75
Permanent Ineff=
       F
Bank Sta=324.6,346.6
XS Rating Curve= 0 ,0
Exp/Cntr(USF)=0,0
Exp/Cntr=0.5,0.3

Type RM Length L Ch R = 1 ,20270.18,53,53.8,55.3
BEGIN DESCRIPTION:
structure xs 3; 12.1 ft between structure and xs
END DESCRIPTION:
XS GIS Cut Line= 6
2220062.61467507463509.4973724182220214.61604646  463288.5345912
2220235.11371962463161.9242048612220229.43445644 463131.82410998
2220235.68164594463094.9088992762220274.17891747462919.600497817
#Sta/Elev= 30
       0 2427.92    10.1  2429.1    53.8 2428.78    63.5 2427.73   107.2 2426.63
   116.9 2424.99   126.6 2426.13   150.9 2425.22   170.3 2425.09     180 2424.56
   191.2 2424.69   218.9 2423.75   238.3  2424.7   262.6 2424.24   303.9 2424.61
   324.3 2422.64   340.32419.068   348.6 2418.33   368.8 2419.13   389.1  2422.2
   413.5 2423.91   429.8 2425.94   462.2 2432.44   503.2 2438.97   535.9 2446.65
   548.2 2448.43   583.9 2452.01   593.3 2452.47   614.1 2452.08     644 2449.78
#Mann= 3 ,-1,0
       0     .05       0   340.3    .045       0   368.8      .1       0
#XS Ineff= 4 ,-1
       0   71.77  2420.5   71.77  252.79 2426.31  252.79     328  2420.5
     381     644    2421
Permanent Ineff=
       F       F       F       F
Bank Sta=340.3,368.8
XS Rating Curve= 0 ,0
Exp/Cntr(USF)=0,0
Exp/Cntr=0.5,0.3

Type RM Length L Ch R = 1 ,20216   ,59.5,58.8,58.9
BEGIN DESCRIPTION:
structure xs 2; 25.2 ft between structure and xs
END DESCRIPTION:
XS GIS Cut Line= 3
2220082.32474667463522.4103954692220266.21842347463282.622175924
2220331.08708238462990.053178417
#Sta/Elev= 30
       0 2428.42     5.1 2428.19    11.6 2427.14    30.7 2426.89    62.2 2425.16
   162.9 2422.43   193.1 2423.72   218.3 2422.96   258.6 2423.26   270.4 2422.57
   290.3  2423.6     316 2421.41   328.5 2421.66   336.4 2419.88   348.7 2419.98
   352.8 2419.47   359.4 2417.78   369.2 2417.06   382.2 2417.73     402 2421.49
   430.7 2421.81   438.9 2422.72   479.8 2421.46     488 2422.18   500.3  2426.9
   514.5 2430.37   533.1  2437.2   557.7 2444.66   578.2 2447.91   601.9 2450.05
#Mann= 4 ,-1,0
       0     .05       0   359.4    .045       0   382.2     .05       0
  392.18      .1       0
#XS Ineff= 6 ,-1
       0   56.79  2420.5   56.79   287.1    2425   287.1     333  2420.5
   407.5   441.3  2420.7   441.3  535.55    2425  535.55   601.9  2420.7
Permanent Ineff=
       F       F       F       F       F       F
Bank Sta=359.4,382.2
XS Rating Curve= 0 ,0
Exp/Cntr(USF)=0,0
Exp/Cntr=0.5,0.3

Type RM Length L Ch R = 1 ,20158   ,156.3,154.6,152.8
BEGIN DESCRIPTION:
structure xs 1
END DESCRIPTION:
XS GIS Cut Line= 3
2220106.10557154463520.7926228122220329.79842442463279.240924003
2220367.10617053  463035.7169664
#Sta/Elev= 30
       0  2427.1    20.7 2426.36    48.5 2426.45    66.3  2425.5   100.3 2425.22
   117.2 2424.38   139.9 2424.62   179.4 2422.84   195.7  2421.2   217.5 2422.33
   267.3 2420.87   284.2 2421.48   315.7 2420.37   335.4 2420.82   343.4 2417.53
   355.6 2417.16   365.5 2415.19   375.2 2414.43   380.32415.185     388 2421.11
   396.1 2421.54   408.2 2420.05   456.8 2420.99   485.1 2418.47   505.3  2418.3
   513.4 2418.99   521.5 2421.88     562 2440.24   570.1 2442.94   575.6 2444.07
#Mann= 4 ,-1,0
       0     .05       0  329.22      .1       0   365.5    .045       0
   380.3      .1       0
#XS Ineff= 2 , 0
             320 2426.05     450            2426
Permanent Ineff=
       F       F
Bank Sta=365.5,380.3
XS Rating Curve= 0 ,0
Exp/Cntr(USF)=0,0
Exp/Cntr=0.3,0.1

Type RM Length L Ch R = 1 ,20003   ,293,290.9,289.1
XS GIS Cut Line= 3
 2220424.2810778463579.6056122632220476.63233414463417.959627749
2220490.40898055463014.763109555
#Sta/Elev= 30
       0 2427.98    19.4 2426.57    55.8 2418.72    65.6  2417.4    99.3 2416.67
   109.8 2417.24   132.9 2415.91   160.6 2415.99     178 2417.05   202.7 2416.34
   218.7 2413.92   242.7 2416.18   282.8 2417.15   290.8 2410.86   298.8 2409.93
   316.2 2410.95   330.8 2413.54   338.8 2416.82   346.8 2417.57   374.8 2417.65
   394.7  2415.9   418.8 2416.14   430.8 2414.25   482.9 2416.72   510.9 2414.56
   518.9 2416.77   534.9 2429.05   546.9 2435.92   562.9  2440.2   573.3 2439.87
#Mann= 4 ,-1,0
       0     .05       0  189.91      .1       0   290.8    .045       0
   316.2      .1       0
#XS Ineff= 2 , 0
             180    2420     500            2420
Permanent Ineff=
       F       F
Bank Sta=290.8,316.2
XS Rating Curve= 0 ,0
Exp/Cntr(USF)=0,0
Exp/Cntr=0.3,0.1

Type RM Length L Ch R = 1 ,19712   ,311.2,309.4,304
XS GIS Cut Line= 5
2220778.04687519463541.037616537  2220805.916864 463487.89727188
 2220774.7766931463308.803951073 2220753.3679649463064.392729256
2220633.29934928463043.638999775
#Sta/Elev= 30
       0 2432.29    49.5 2430.08    70.8 2427.51   103.4 2420.25   122.7 2417.46
   131.8 2413.75     144 2407.11     148 2406.02   160.2 2404.86   204.9 2408.62
   245.4 2408.83   265.92407.896   281.6 2407.28   291.7 2407.88   301.6 2409.25
   317.7 2408.47   333.8 2408.84   369.9 2407.21     394 2409.12     410 2407.07
   446.2 2408.01   458.2 2407.62   462.3 2408.06   470.3 2411.68   476.2 2415.66
   482.3 2421.59   486.3 2424.25   532.5  2430.8   565.5 2434.52     609 2436.88
#Mann= 3 ,-1,0
       0      .1       0   265.9    .045       0   291.7      .1       0
Bank Sta=265.9,291.7
XS Rating Curve= 0 ,0
Exp/Cntr(USF)=0,0
Exp/Cntr=0.3,0.1

Type RM Length L Ch R = 1 ,19403   ,132.2,131.6,131.2
XS GIS Cut Line= 4
2221082.80477607463338.9735216792221084.64166226463245.292326108
2221005.65555619463142.4266995982220954.22274294462953.227422268
#Sta/Elev= 30
       0 2408.47    45.8 2407.14    53.8 2407.44    69.8 2406.41    81.8  2405.1
    93.7 2402.58   122.6 2402.48   134.2 2399.18     147 2400.57   173.3 2401.32
   186.4  2400.8   199.6 2401.75   216.8 2401.86   228.9 2400.91   238.7 2401.88
   253.7 2401.79   274.4 2400.25     281 2397.09   287.5 2396.07   303.4 2397.14
     320 2400.08   329.9 2404.26   339.7 2411.25   357.3  2426.7   365.6 2431.15
   375.5 2434.37   390.5 2437.31   399.5 2440.73   411.4 2443.93   419.5 2447.71
#Mann= 4 ,-1,0
       0     .05       0      40      .1       0     281    .045       0
   303.4      .1       0
#XS Ineff= 2 , 0
             120    2408
Permanent Ineff=
       F       F
Bank Sta=281,303.4
XS Rating Curve= 0 ,0
Exp/Cntr(USF)=0,0
Exp/Cntr=0.3,0.1

Type RM Length L Ch R = 1 ,19271   ,259,249.6,244.7
XS GIS Cut Line= 3
2221106.92844118463336.9539025982221146.41835102463145.875263865
2221066.85414547462889.449836468
#Sta/Elev= 30
       0 2407.97      57 2406.32    77.4 2404.01    89.6 2401.21    93.7 2401.02
   134.6 2401.16   146.8 2400.03   163.2 2401.75   171.3 2401.74   204.2 2398.77
   237.7 2399.25   261.4 2397.57   274.2 2395.53  278.652393.932     287 2392.41
   299.7 2392.21   312.5 2393.92   324.2 2394.88   329.9 2397.87   338.2 2400.88
   350.9 2407.94   364.7  2417.8   380.1  2425.9   392.7  2429.1   405.2 2434.65
   426.2 2441.25   434.6 2442.55   442.9 2441.93   447.1 2442.71   463.6 2449.13
#Mann= 5 ,-1,0
       0     .05       0      40     .06       0     140      .1       0
  278.65    .045       0   312.5      .1       0
Bank Sta=278.65,312.5
XS Rating Curve= 0 ,0
Exp/Cntr(USF)=0,0
Exp/Cntr=0.3,0.1

Type RM Length L Ch R = 1 ,19021   ,271.6,267.9,262.3
XS GIS Cut Line= 3
2221540.14831744463162.3420581322221365.68524898462950.472092987
2221208.63147993462781.478563721
#Sta/Elev= 30
       0 2420.38      15 2418.27    22.2 2416.14      44 2403.96    63.3 2394.96
    75.5 2391.76    94.8 2393.12   120.7 2392.52   146.6 2394.22   174.1 2393.43
   198.4 2393.63   213.9 2392.66   250.9 2394.19   282.1  2392.3   335.4 2393.22
   347.5 2388.68   352.9 2387.84   364.2 2387.56   372.7 2387.77   376.6 2388.64
   386.8 2394.57   401.8 2408.56   405.9 2411.59     418 2416.94   429.4 2425.53
   435.3  2428.9     440 2430.88   447.1 2432.64   494.1 2450.37   505.2 2455.33
#Mann= 5 ,-1,0
       0      .1       0      60     .05       0     210      .1       0
   347.5    .045       0   376.6      .1       0
#XS Ineff= 2 , 0
             250    2400
Permanent Ineff=
       F       F
Bank Sta=347.5,376.6
XS Rating Curve= 0 ,0
Exp/Cntr(USF)=0,0
Exp/Cntr=0.3,0.1

Type RM Length L Ch R = 1 ,18754   ,245.6,244.8,242.3
XS GIS Cut Line= 4
2221683.60593378463008.7658919862221633.02472887462916.349601621
2221598.35091799462772.042906796 2221367.9895689 462599.30044544
#Sta/Elev= 30
       0 2418.45     8.6 2416.88      17 2413.56    58.8 2389.41    63.4 2387.31
    67.9 2386.28      77 2387.01    90.7  2390.1    99.5  2390.4   149.8  2386.4
   178.5 2386.25   199.1 2387.69     232 2388.46   291.5 2388.62   326.5 2386.66
   334.5  2385.5   374.5 2387.04   383.42385.309   388.8  2384.1   397.4  2383.8
     4412385.399   443.1 2386.81   451.5 2395.68   465.2 2407.59   474.5 2413.37
   491.5 2422.45   496.5 2423.81   506.5 2424.34   518.6 2427.82   541.7 2430.62
#Mann= 3 ,-1,0
       0      .1       0   383.4    .045       0     441      .1       0
#XS Ineff= 2 , 0
          260.96 2394.21
Permanent Ineff=
       F       F
Bank Sta=383.4,441
XS Rating Curve= 0 ,0
Exp/Cntr(USF)=0,0
Exp/Cntr=0.3,0.1

Type RM Length L Ch R = 1 ,18509   ,284.2,295.4,311.4
XS GIS Cut Line= 2
2221910.32200362462683.2051526812221516.30991636    462412.26444
#Sta/Elev= 30
       0 2403.01     7.5 2400.49    31.7 2388.73    38.9  2386.5      56 2377.73
    60.5 2375.99    65.7 2375.31    88.3 2376.99    95.3 2378.73   116.5 2376.43
   126.7 2377.34   144.8 2377.45   194.2 2380.77   287.8 2382.12   300.1  2382.9
   339.5  2381.7   347.3 2380.66   353.9 2377.99     357 2376.57   368.3  2376.2
   376.4 2376.43   380.32377.927   386.1 2384.49   391.3 2389.45   398.9 2395.06
   424.9 2408.99   434.2 2411.83   449.2 2414.74   463.8 2415.06   478.2  2416.7
#Mann= 3 ,-1,0
       0      .1       0   353.9    .045       0   380.3      .1       0
Bank Sta=353.9,380.3
XS Rating Curve= 0 ,0
Exp/Cntr(USF)=0,0
Exp/Cntr=0.3,0.1

Type RM Length L Ch R = 1 ,18213   ,323.7,329,331.1
XS GIS Cut Line= 4
2221972.61095675462621.5879043322221894.12787514 462516.08530513
2221877.57772211462390.238638992 2221799.1795447462192.936559157
#Sta/Elev= 30
       0 2404.07    20.8 2399.19    34.2 2394.54    45.4 2388.59    55.3 2382.19
    74.4 2372.08    80.6 2370.63   103.5 2374.61   134.4 2377.08   146.5 2376.97
   182.8 2374.09   194.9 2374.72     203 2376.66     207 2377.06   289.7 2377.74
   315.5 2376.75   319.8 2375.48   328.4 2374.12   332.8 2372.73     338 2371.68
   354.3 2371.89   359.82372.679   377.4 2377.41   401.6 2377.93   414.5 2376.75
     436 2376.65   440.3 2377.39   448.9 2380.12   461.9 2381.96   470.7 2385.27
#Mann= 3 ,-1,0
       0      .1       0   332.8    .045       0   359.8      .1       0
#XS Ineff= 1 ,-1
  134.08  251.83 2379.13
Permanent Ineff=
       F
Bank Sta=332.8,359.8
XS Rating Curve= 0 ,0
Exp/Cntr(USF)=0,0
Exp/Cntr=0.3,0.1

Type RM Length L Ch R = 1 ,17884   ,492.8,477.4,460.9
XS GIS Cut Line= 4
2222307.85068161462383.8376633182222152.79098039462237.760252172
2222114.55586443462027.9527393942221959.62366242461971.579224189
#Sta/Elev= 30
       0  2419.6    52.6 2415.58    72.4 2412.41    89.4 2407.82    92.2 2406.34
    97.9 2400.81     104 2389.49   108.9 2378.02     112 2374.31   114.8 2371.57
   123.3 2367.22   132.2 2365.24   221.8 2370.29   263.7 2366.97   279.4 2365.73
   290.9 2366.93   294.9 2369.24   307.1 2369.44   319.3 2372.92   347.8 2373.94
   433.1 2370.86   467.8 2372.15   475.6 2371.76   488.4 2368.87     499 2368.38
   520.8 2374.11   552.3 2377.74   564.5 2380.16     577 2385.42   591.2 2394.14
#Mann= 3 ,-1,0
       0      .1       0   263.7    .045       0   290.9      .1       0
#XS Ineff= 1 ,-1
  436.39   557.8 2380.31
Permanent Ineff=
       F
Bank Sta=263.7,290.9
XS Rating Curve= 0 ,0
Exp/Cntr(USF)=0,0
Exp/Cntr=0.3,0.1

Type RM Length L Ch R = 1 ,17407   ,172.7,174.4,176.4
XS GIS Cut Line= 2
2222556.66582118461999.3259844482222123.15408133461707.286258671
#Sta/Elev= 30
       0 2410.59      11 2405.02    19.2 2399.29    24.7 2393.91    29.5 2388.32
    39.2 2375.96      44 2372.36    56.7 2360.95    61.1 2358.79    68.42358.201
    82.6 2356.78   101.52358.078   106.7 2360.52   116.3 2361.08   169.4  2359.3
     179 2360.03   193.5 2358.89   223.8 2359.69   238.2 2358.45   254.4 2359.28
   299.6 2359.18   314.1 2359.88   328.6 2361.94   347.7 2363.31   362.3 2365.83
   420.2  2370.4     454 2375.28   477.4  2380.9   502.2 2388.99   522.7 2397.57
#Mann= 3 ,-1,0
       0      .1       0    68.4    .045       0   101.5      .1       0
Bank Sta=68.4,101.5
XS Rating Curve= 0 ,0
Exp/Cntr(USF)=0,0
Exp/Cntr=0.3,0.1

Type RM Length L Ch R = 1 ,17233   ,423.4,422,415.5
XS GIS Cut Line= 2
2222664.99235311461879.1373860642222310.38147458 461575.77563217
#Sta/Elev= 30
       0 2397.68    13.3 2395.97    22.1 2392.61    27.4 2389.23    32.7 2384.36
    38.8  2376.6    43.2 2372.27      53 2364.98    58.4 2362.17    64.2 2360.79
      83 2359.21    92.8 2356.26   104.1 2355.96   135.3 2356.03   169.5  2355.7
   193.8 2357.88   273.8 2354.78   285.7 2355.52   295.9 2358.47   299.9 2358.98
   311.7 2356.83   343.2 2354.65   374.8  2356.1   393.5 2356.11   406.4 2355.17
   415.3 2355.55   422.2 2358.01   430.4 2361.88   453.1 2369.58   466.7 2377.63
#Mann= 3 ,-1,0
       0      .1       0   104.1    .045       0   135.3      .1       0
Bank Sta=104.1,135.3
XS Rating Curve= 0 ,0
Exp/Cntr(USF)=0,0
Exp/Cntr=0.3,0.1

Type RM Length L Ch R = 1 ,16811   ,319.4,322.6,325.9
XS GIS Cut Line= 2
2222826.17243885461728.1107420172222445.34990131461332.432223119
#Sta/Elev= 30
       0 2410.21    20.7 2395.59    31.8 2392.84    42.9 2382.84    62.9  2366.4
    70.7 2360.84    76.2 2357.83    82.7 2356.23    91.2  2355.8     104 2353.85
   141.3 2353.55   176.1 2352.11   204.8 2352.53   227.8 2350.79   250.9 2353.18
   269.4 2352.31   303.4 2352.23   331.7 2350.62   362.8 2350.95   389.4 2349.82
   406.7 2350.28   413.7  2349.8   422.2 2347.74   433.5  2347.1   453.8 2347.83
   464.9 2351.21   470.3 2353.93   509.3 2388.88   531.5 2405.07   549.2 2416.72
#Mann= 3 ,-1,0
       0      .1       0   422.2    .045       0   453.8      .1       0
#XS Ineff= 2 , 0
          251.49 2358.08
Permanent Ineff=
       F       F
Bank Sta=422.2,453.8
XS Rating Curve= 0 ,0
Exp/Cntr(USF)=0,0
Exp/Cntr=0.3,0.1

Type RM Length L Ch R = 1 ,16488   ,333.5,332.9,332.8
XS GIS Cut Line= 4
 2222891.0706759461554.2451951392222776.44925841461319.638193589
2222794.91981383461253.6719242282222699.61690697461099.167782304
#Sta/Elev= 30
       0 2369.66     8.9 2363.56    24.8 2354.58    33.9 2351.72    45.7 2350.11
    54.6 2349.59    92.7 2350.31     108 2349.58   121.4  2350.5   143.5 2350.31
     198 2346.71   233.2 2346.91   254.9 2348.04   305.1 2346.84     349  2345.2
   352.3 2343.63   358.1 2339.48   363.9 2338.54   380.5 2339.46   391.3    2340
   400.7 2343.41   414.8 2342.48   418.7 2344.01   428.9 2352.53   438.3 2361.45
   456.7 2381.45   466.5 2389.34   479.6 2398.45   504.1 2409.78   511.1 2412.47
#Mann= 3 ,-1,0
       0      .1       0   358.1    .045       0   380.5      .1       0
Bank Sta=358.1,380.5
XS Rating Curve= 0 ,0
Exp/Cntr(USF)=0,0
Exp/Cntr=0.3,0.1

Type RM Length L Ch R = 1 ,16155   ,324,323.9,324.4
XS GIS Cut Line= 2
2223209.04010193461275.6778833672222990.83184145460952.938719663
#Sta/Elev= 30
       0    2372    16.8 2361.71      23 2356.78    28.3 2354.78      37 2353.02
    48.5 2347.27    54.3 2345.23      60 2344.12      73  2343.5     109 2343.79
   123.4  2341.8   137.8  2342.6   158.7  2341.8   186.5 2342.73   225.1 2340.85
   250.2 2341.29   265.8 2337.51   276.1 2338.17   292.7 2337.61     312 2338.68
   319.3 2334.42   322.9 2333.46   336.2 2333.21   347.1 2334.41   356.8 2337.38
   368.3 2344.03   374.8 2346.73   379.8 2350.51   384.5 2355.33   389.6 2359.07
#Mann= 3 ,-1,0
       0      .1       0   319.3    .045       0   347.1      .1       0
Bank Sta=319.3,347.1
XS Rating Curve= 0 ,0
Exp/Cntr(USF)=0,0
Exp/Cntr=0.3,0.1

Type RM Length L Ch R = 1 ,15831   ,78.9,81.4,86
XS GIS Cut Line= 2
2223448.60800077461045.9258113372223235.34551438460739.257662306
#Sta/Elev= 30
       0 2371.77     7.8 2370.94    14.8 2368.31    20.4 2364.22    23.8  2362.3
    32.5 2358.74    49.6 2348.21    61.2 2342.74      74 2339.41    84.8 2338.09
   101.4 2333.97   127.3 2333.14   147.1 2334.33   181.2 2333.22   195.8 2334.29
     225 2333.38     260 2333.48     264 2333.13   273.7  2331.2   278.6 2329.34
   282.5 2328.73     288 2328.66   305.5 2329.26     309 2330.23   314.1  2333.8
     317  2336.4     323 2342.79   342.8 2359.66   351.4 2365.56   373.5 2378.12
#Mann= 3 ,-1,0
       0      .1       0   278.6    .045       0   305.5      .1       0
Bank Sta=278.6,305.5
XS Rating Curve= 0 ,0
Exp/Cntr(USF)=0,0
Exp/Cntr=0.3,0.1

Type RM Length L Ch R = 1 ,15750   ,102.7,102.9,99.4
BEGIN DESCRIPTION:
structure xs 4
END DESCRIPTION:
XS GIS Cut Line= 2
2223466.44745112460986.911263211 2223307.0378237460681.158371281
#Sta/Elev= 30
       0 2352.58       3 2351.19    14.8  2343.9      29 2336.48      38 2333.32
    44.5 2332.13    60.6 2331.57    74.1    2333      86 2333.03   123.8  2332.3
   150.8 2333.37   168.9 2332.37   195.9 2332.23   203.9 2332.46     223 2331.29
   236.5 2331.39     241 2330.78   246.1 2328.82   250.1 2327.83   260.9 2327.58
   290.4 2328.62   290.9 2329.05   295.2 2335.02   304.2 2348.77   308.7 2354.12
   313.2 2357.62   323.2 2364.25   332.1 2371.11   335.8 2373.39   344.8 2378.17
#Mann= 5 ,-1,0
       0      .1       0      60     .06       0     170      .1       0
   246.1    .045       0   290.9      .1       0
#XS Ineff= 1 ,-1
   17.15  151.24 2336.05
Permanent Ineff=
       F
Bank Sta=246.1,290.9
XS Rating Curve= 0 ,0
Exp/Cntr(USF)=0,0
Exp/Cntr=0.5,0.3

Type RM Length L Ch R = 1 ,15647   ,73.4,75.2,73
BEGIN DESCRIPTION:
structure xs 3; 25.7 ft between structure and xs
END DESCRIPTION:
XS GIS Cut Line= 4
2223419.47959676461211.400458651 2223540.2409891460912.667210955
2223392.91760333460638.3896109952223291.83823168460652.543102122
#Sta/Elev= 30
       0  2376.2    32.6 2372.49    62.8  2370.1   105.9 2364.75   151.3 2361.03
   222.4 2353.25   235.4  2350.7     244 2346.65   251.1 2347.05   257.3 2346.31
     288 2333.92   300.1 2330.57   304.4 2330.05   507.8 2331.85   521.4 2329.29
   534.6 2330.04   561.2 2329.61   566.8 2328.47571.37812326.349   575.9 2325.41
   584.4 2325.19   596.6 2325.43604.15512326.404   609.8 2328.54   626.1 2341.47
   654.6 2356.99   666.6 2362.74   678.7 2370.49   707.5 2383.32   735.6 2392.79
#Mann= 7 ,-1,0
       0      .1       0     300     .06       0  472.22      .1       0
  522.22     .06       0571.3781    .045       0604.1551     .06       0
  653.56      .1       0
#XS Ineff= 4 ,-1
       0   46.99  2326.9   46.99     500 2336.51     500     546  2326.9
     630     700  2329.2
Permanent Ineff=
       F       F       F       F
Bank Sta=571.3781,604.1551
XS Rating Curve= 0 ,0
Exp/Cntr(USF)=0,0
Exp/Cntr=0.5,0.3

Type RM Length L Ch R = 1 ,15572   ,59.4,55.9,53.6
BEGIN DESCRIPTION:
structure xs 2; 23.6 ft between structure and xs
END DESCRIPTION:
XS GIS Cut Line= 6
 2223840.3941262461158.1930398992223550.69010259460872.004492567
2223511.25503537460800.849914751 2223504.3967628460697.975826342
2223448.16479896 460593.620331782223357.68468064460588.334596904
#Sta/Elev= 30
       0 2422.39      33 2414.27      66 2403.54   122.6 2382.28   185.3 2355.45
   218.8 2343.92   244.3 2337.65   252.8 2333.31     267 2333.28   332.1 2329.19
     342 2327.48   354.9 2329.24   429.9 2329.84   513.4 2331.79   573.5  2331.3
   592.7 2330.19   618.5 2330.76   646.6 2329.05656.34952325.903   666.3 2324.29
   679.1 2324.04     686 2324.37690.94272325.824   698.2 2329.98   719.3 2331.66
   735.3 2336.69   771.4  2337.9   779.4 2342.02   787.4 2349.24   801.9 2356.56
#Mann= 7 ,-1,0
       0      .1       0     180     .06       0     330     .05       0
  373.53     .06       0656.3495    .045       0690.9427     .06       0
  791.28      .1       0
#XS Ineff= 3 ,-1
   33.13     410 2334.89     410     648  2326.9     699   801.9  2328.4
Permanent Ineff=
       F       F       F
Bank Sta=656.3495,690.9427
XS Rating Curve= 0 ,0
Exp/Cntr(USF)=0,0
Exp/Cntr=0.5,0.3

Type RM Length L Ch R = 1 ,15516   ,117.4,119.2,121.4
BEGIN DESCRIPTION:
structure xs 1
END DESCRIPTION:
XS GIS Cut Line= 2
  2223766.021934 460936.814771792223470.92616795460539.220756469
#Sta/Elev= 30
       0 2356.31    16.5 2347.66    35.4 2339.25    38.2 2337.39    43.4 2332.61
    49.7 2327.72    52.5 2327.12    69.7 2327.02    72.5 2326.36    79.2 2323.24
    95.4 2324.93   124.1 2326.41   203.8 2327.36   243.6 2328.61   271.6 2328.13
   304.1 2329.08   361.3 2327.23   389.9 2328.18   398.5 2329.66     403 2329.94
   407.1 2329.09   416.72325.209   424.2 2323.95   438.5 2323.88   447.9 2324.06
   452.8 2325.22   452.8 2325.23   464.3 2327.54   472.8 2327.94   495.1 2336.65
#Mann= 9 ,-1,0
       0     .06       0     130     .05       0     170     .08       0
     250     .05       0     330     .06       0     370      .1       0
   416.7    .045       0   452.8      .1       0  495.14     .06       0
#XS Ineff= 2 , 0
          401.16 2333.76
Permanent Ineff=
       F       F
Bank Sta=416.7,452.8
XS Rating Curve= 0 ,0
Exp/Cntr(USF)=0,0
Exp/Cntr=0.3,0.1

Type RM Length L Ch R = 1 ,15397   ,134.9,150.4,159.9
XS GIS Cut Line= 2
2223829.18179178460854.1730356312223553.96395658460445.725012554
#Sta/Elev= 30
       0 2337.84     4.3 2334.47    10.8 2328.25    15.8 2325.66    30.3 2325.31
      35 2324.72    44.6 2322.22    59.1 2321.34    67.7  2322.6   112.1 2323.62
     117 2324.35   126.6 2326.78   130.7 2326.98   141.1 2325.44   150.7 2324.82
   218.2  2324.5   256.8 2325.47   266.5 2325.15   358.1 2325.98   370.3 2327.63
   373.2 2327.44   384.32323.827   387.6 2323.43   420.8 2323.23   428.8 2323.76
   445.6 2325.41   453.9 2330.99   464.2 2339.48   473.9 2345.62   492.5 2359.69
#Mann= 7 ,-1,0
       0     .06       0      20      .1       0     110     .05       0
     260     .06       0     290      .1       0   384.3    .045       0
   428.8      .1       0
#XS Ineff= 2 , 0
          367.94 2330.93
Permanent Ineff=
       F       F
Bank Sta=384.3,428.8
XS Rating Curve= 0 ,0
Exp/Cntr(USF)=0,0
Exp/Cntr=0.3,0.1

Type RM Length L Ch R = 1 ,15246   ,307.7,323.3,298
XS GIS Cut Line= 4
2223957.33749847460800.0389168382223739.15188346460485.787593637
2223735.43777898460436.7225071972223627.30434473460314.948879596
#Sta/Elev= 30
       0 2345.74     9.1 2341.68      23 2331.47    28.8 2325.55    32.7 2322.96
    47.3 2322.54    61.9 2320.02    76.5 2318.79      96 2320.43   120.4 2320.12
   173.9 2321.81   186.8  2323.5   212.9  2324.4     320 2324.74   349.2 2324.61
   368.7 2323.03   383.2 2324.02   395.2 2321.76   400.8 2321.58   427.7 2321.57
   459.3 2323.05   484.7 2321.34   495.4 2324.64     521 2329.47   544.3    2341
   551.1 2345.41   563.2 2349.74   569.2 2353.68   581.3 2358.92   594.6 2366.78
#Mann= 5 ,-1,0
       0     .06       0     200     .07       0     320      .1       0
   400.8    .045       0   427.7      .1       0
#XS Ineff= 2 , 0
          382.72  2332.1  510.47         2329.38
Permanent Ineff=
       F       F
Bank Sta=400.8,427.7
XS Rating Curve= 0 ,0
Exp/Cntr(USF)=0,0
Exp/Cntr=0.3,0.1

Type RM Length L Ch R = 1 ,14923   ,366.9,379.9,361
XS GIS Cut Line= 3
2224178.14424054460679.2808903092224054.09872095460484.024053922
2223891.00183408460095.807520399
#Sta/Elev= 30
       0 2364.16      12 2357.93    26.2  2348.1    43.5 2334.02      58 2319.43
    63.8 2317.11    78.3 2317.06    92.5 2314.03     102 2316.17   111.5 2316.65
   150.7 2318.01   206.3 2317.03   234.4 2319.01   247.4 2318.08   260.4  2315.4
   295.2  2314.3   303.8 2313.62  309.67 2314.33   321.2  2317.5   347.2 2318.31
   368.9 2317.17   412.2 2321.18   425.3 2320.74   442.7 2318.06   470.2 2319.37
   585.8 2320.01   598.9 2321.76   607.7 2324.94   632.1 2339.11   652.4 2348.78
#Mann= 5 ,-1,0
       0      .1       0      30     .06       0     160      .1       0
   295.2    .045       0  309.67      .1       0
#XS Ineff= 2 , 0
                             400            2325
Permanent Ineff=
       F       F
Bank Sta=295.2,309.67
XS Rating Curve= 0 ,0
Exp/Cntr(USF)=0,0
Exp/Cntr=0.3,0.1

Type RM Length L Ch R = 1 ,14543   ,383.3,386.2,387.4
XS GIS Cut Line= 2
2224472.65739204460456.5341574092224111.73645493460034.302591465
#Sta/Elev= 30
       0 2345.52     4.4 2340.91    13.1 2330.53    16.9 2327.19    25.4 2318.44
    30.7 2314.26    59.5 2312.45    80.8 2309.34    88.6 2309.84   121.9 2308.49
   133.2 2308.17   136.2 2308.44   146.5 2310.14   161.6 2310.59   183.3 2310.11
   188.6 2309.56   204.4 2310.99   229.7 2311.12   255.2 2309.94   266.6 2312.14
   296.2 2312.65   320.9 2311.71   374.4 2313.55   408.4 2314.03   419.4  2315.1
   435.9 2312.96   462.2 2311.84     478  2313.5   493.5 2314.43   555.5 2315.75
#Mann= 4 ,-1,0
       0     .06       0    30.7      .1       0   121.9    .045       0
   136.2      .1       0
#XS Ineff= 2 , 0
                             300            2315
Permanent Ineff=
       F       F
Bank Sta=121.9,136.2
XS Rating Curve= 0 ,0
Exp/Cntr(USF)=0,0
Exp/Cntr=0.3,0.1

Type RM Length L Ch R = 1 ,14157   ,614.4,624.3,626.1
XS GIS Cut Line= 3
2224777.21408758460300.9272108032224538.96500615459878.103145954
2224280.48185997 459718.16742533
#Sta/Elev= 30
       0 2378.78    13.5 2368.36    31.9  2351.5    54.8 2327.61    73.2 2306.54
    77.8 2304.58    96.1 2304.18   105.62300.321   114.5 2299.36   128.3 2300.35
   138.6 2302.91     188 2303.29   201.7  2305.2   220.1  2302.1   238.4 2301.28
     266 2301.88   275.2 2303.28   285.4 2301.55   316.5 2302.54   353.2 2301.23
   385.4  2303.2   420.5 2302.22   473.4 2306.16   557.8 2306.83   643.8  2309.3
   688.5 2312.23   723.8 2312.01     738 2316.23   766.1 2327.01   789.3 2337.67
#Mann= 5 ,-1,0
       0      .1       0      50     .06       0   105.6    .045       0
   128.3     .06       0     180      .1       0
Bank Sta=105.6,128.3
XS Rating Curve= 0 ,0
Exp/Cntr(USF)=0,0
Exp/Cntr=0.3,0.1

Type RM Length L Ch R = 1 ,13532   ,335.1,340,344.9
XS GIS Cut Line= 2
2225029.33047699460179.7052897142224980.89855683459598.003494402
#Sta/Elev= 30
       0 2316.61    10.6 2309.25    22.6 2298.93    26.6  2297.8    42.7  2297.6
    54.7 2294.05    62.7 2295.25    90.8 2296.96     127 2295.58     143 2296.97
   187.2 2297.65   251.4 2295.15   279.5  2292.6   299.6 2293.24   339.7 2291.83
   351.8 2293.16   371.8 2292.89   383.8 2291.92   403.6 2292.16     416 2291.12
   422.42288.862     432 2287.67   449.62288.932   464.1 2292.52   476.2 2293.34
   480.2 2294.37   522.2 2308.47   529.6  2311.5   560.5 2326.86   583.7 2340.52
#Mann= 4 ,-1,0
       0     .06       0      30      .1       0   422.4    .045       0
   449.6      .1       0
#XS Ineff= 2 , 0
             300    2295
Permanent Ineff=
       F       F
Bank Sta=422.4,449.6
XS Rating Curve= 0 ,0
Exp/Cntr(USF)=0,0
Exp/Cntr=0.3,0.1

Type RM Length L Ch R = 1 ,13193   ,293,293.1,293.2
XS GIS Cut Line= 2
2225244.72157281460187.7887506172225348.00370915459622.782976138
#Sta/Elev= 30
       0 2297.96    10.8 2293.48      19 2292.15    55.5  2290.5    63.6 2291.38
   100.2 2288.75   116.5 2290.98   132.8 2291.44   165.3 2289.09   189.7 2290.25
   201.9 2289.04   218.2 2290.69   246.6 2288.68   266.5 2289.35   283.2 2287.25
   315.8 2286.52   352.4 2287.89   373.1 2286.13     393 2287.14   433.7  2285.4
   447.92281.099     454 2279.16   470.3 2279.39     4782281.165   483.1 2283.32
   496.8 2299.02   523.1  2320.6   531.3 2326.05   556.2 2346.46   574.4 2357.21
#Mann= 5 ,-1,0
       0      .1       0      40     .06       0     140      .1       0
   447.9    .045       0     478      .1       0
Bank Sta=447.9,478
XS Rating Curve= 0 ,0
Exp/Cntr(USF)=0,0
Exp/Cntr=0.3,0.1

Type RM Length L Ch R = 1 ,12899   ,320.4,318.2,317.2
XS GIS Cut Line= 2
2225524.89938315460247.3114776912225636.77032931459665.901973718
#Sta/Elev= 30
       0 2293.56     6.2 2291.65    14.4 2290.42    59.2 2288.66   173.3 2287.32
   201.8 2286.21   230.3 2286.78   254.7 2281.67   287.3 2281.34   305.2 2282.35
   319.9 2279.36     324 2279.17   336.2 2281.29   368.8 2279.81   409.5  2279.9
   442.1 2278.57   454.3  2276.2   464.52275.632   486.9 2274.47   491.42275.557
     495  2278.3   502.9 2286.54   515.4 2294.26   520.4 2298.97   531.7 2307.87
   548.3 2326.58   567.8 2343.55   580.6 2356.24   584.7 2359.26   592.1 2363.14
#Mann= 5 ,-1,0
       0      .1       0     100     .06       0     200      .1       0
   464.5    .045       0   491.4      .1       0
#XS Ineff= 2 , 0
             420    2285
Permanent Ineff=
       F       F
Bank Sta=464.5,491.4
XS Rating Curve= 0 ,0
Exp/Cntr(USF)=0,0
Exp/Cntr=0.3,0.1

Type RM Length L Ch R = 1 ,12581   ,327.5,319.2,312.3
XS GIS Cut Line= 2
2225891.16933215460188.6068589212225937.29667608459726.007243072
#Sta/Elev= 30
       0    2281    95.9 2280.58   103.9 2280.06     120 2280.87   168.3 2278.03
   208.5  2278.1   212.5 2277.81   220.5 2275.37   228.6  2273.8   240.6 2273.19
   252.7 2274.16   256.7 2273.33   260.7  2271.5   264.7 2270.88   272.8 2271.36
   280.8 2274.99   301.9 2274.79     309 2273.98     317  2271.3   324.2 2269.85
   336.7 2269.06   349.92269.833   362.3 2272.22   389.3  2273.4   393.4 2274.59
   401.4 2281.77   409.4 2291.26   429.5 2312.02   458.1 2338.52   464.9 2343.76
#Mann= 5 ,-1,0
       0     .05       0      40     .06       0     240      .1       0
   324.2    .045       0   349.9      .1       0
#XS Ineff= 2 , 0
             300    2280
Permanent Ineff=
       F       F
Bank Sta=324.2,349.9
XS Rating Curve= 0 ,0
Exp/Cntr(USF)=0,0
Exp/Cntr=0.3,0.1

Type RM Length L Ch R = 1 ,12262   ,413.3,402.6,393.1
XS GIS Cut Line= 4
2226294.69940274460079.4670890822226310.71920277460012.582051227
2226256.40629453459871.4794167262226171.32975385459651.238610904
#Sta/Elev= 30
       0 2274.03    59.9  2274.2      64 2274.04    72.4 2272.27    89.6  2272.2
    98.1 2273.56   123.9 2274.04   192.4 2270.02   220.6 2269.99   235.3 2269.08
   248.2 2269.39   276.1 2267.62     291 2267.43   320.9 2268.19   336.4 2267.26
   339.5 2266.34   342.6 2264.12   351.1  2263.2   356.3 2264.05   361.1 2264.69
   372.5  2264.8   381.1 2266.67   385.4 2267.03   398.2 2264.94   406.8 2264.86
   411.1 2265.51   415.4 2268.35   419.9 2272.77   447.2  2292.3   456.1 2299.37
#Mann= 4 ,-1,0
       0     .06       0  138.78      .1       0   342.6    .045       0
   356.3      .1       0
#XS Ineff= 2 , 0
          294.02 2274.44
Permanent Ineff=
       F       F
Bank Sta=342.6,356.3
XS Rating Curve= 0 ,0
Exp/Cntr(USF)=0,0
Exp/Cntr=0.3,0.1

Type RM Length L Ch R = 1 ,11859   ,355.8,363,368.7
XS GIS Cut Line= 3
2226571.01527687459874.9637801662226609.07759201459554.568721966
2226365.87337929459395.428261626
#Sta/Elev= 30
       0 2266.76     6.3  2265.9    50.1 2266.56    82.4 2266.25    98.5 2265.88
   122.6 2264.13   142.4 2263.89   151.6 2264.01     171 2265.69   252.1 2265.58
   283.5 2266.76   396.5 2265.42   412.9 2266.09   427.5 2265.67     437 2264.46
   455.92259.227   462.4  2258.2   477.4 2258.19   488.62259.056   500.5 2260.75
   532.3 2260.27   543.9 2261.31   546.8 2263.23   558.4 2274.62   567.5 2282.56
   581.9 2297.28   596.2 2314.67   598.8 2317.18   604.6 2322.16   613.3 2328.08
#Mann= 4 ,-1,0
       0     .06       0     120      .1       0   455.9    .045       0
   488.6      .1       0
Bank Sta=455.9,488.6
XS Rating Curve= 0 ,0
Exp/Cntr(USF)=0,0
Exp/Cntr=0.3,0.1

Type RM Length L Ch R = 1 ,11496   ,89.2,92.4,114.1
BEGIN DESCRIPTION:
structure xs 4
END DESCRIPTION:
XS GIS Cut Line= 3
2226712.13199622459644.9957930732226785.30362848 459280.44426808
2226615.44091074459077.915643083
#Sta/Elev= 30
       0 2262.33    24.3 2262.43    40.5 2261.38    65.1 2260.59    97.7 2260.86
   158.9 2259.92   234.3 2259.59   285.3 2258.47   342.5 2258.31   400.5 2256.26
   417.2 2252.59   440.2 2251.78   445.9 2251.98   449.2 2252.63   454.4 2254.81
   459.6 2255.53   477.2 2254.57   537.9 2256.19   547.9 2256.89   559.5 2256.25
   576.5 2256.61   579.4 2257.69   590.1 2264.92   595.4 2270.26   602.1 2278.76
   604.9 2281.16     611 2285.44   622.6 2293.25   627.6 2295.52   636.2 2298.34
#Mann= 8 ,-1,0
       0      .1       0      50     .06       0     190     .07       0
     290      .1       0  391.82     .06       0   417.2    .045       0
   449.2     .06       0  471.82      .1       0
Bank Sta=417.2,449.2
XS Rating Curve= 0 ,0
Exp/Cntr(USF)=0,0
Exp/Cntr=0.5,0.3

Type RM Length L Ch R = 1 ,11404   ,51.4,51.1,46.2
BEGIN DESCRIPTION:
structure xs 3; 14.5 ft between structure and xs
END DESCRIPTION:
XS GIS Cut Line= 3
2226741.92891883459606.5014896372226831.54732009459224.129644282
2226652.31051758458813.876518537
#Sta/Elev= 30
       0 2261.34   120.5 2258.76   421.8 2255.99   439.6 2254.57   450.52251.274
   457.1 2250.25   491.1 2249.71   505.1  2251.4     516 2254.37   526.9 2255.49
     581 2254.98   588.9 2254.49     598  2252.2   613.2 2251.81   628.4 2252.79
   640.4 2255.25   644.8  2254.7   655.5 2255.46   661.8 2257.05   670.9 2262.98
   683.1 2268.08   701.5 2278.33   710.4 2281.73     719 2283.69   727.7 2284.58
   740.7  2287.9     767 2292.49   797.5 2291.45   822.8 2293.55   840.4 2293.95
#Mann= 9 ,-1,0
       0     .06       0     150     .07       0     250      .1       0
     350     .06       0     360      .1       0  422.73     .06       0
   450.5    .045       0   505.1     .06       0  672.73      .1       0
#XS Ineff= 3 ,-1
       0     435  2250.6   519.5  538.03  2252.7  538.03  699.15 2257.55
Permanent Ineff=
       F       F       F
Bank Sta=450.5,505.1
XS Rating Curve= 0 ,0
Exp/Cntr(USF)=0,0
Exp/Cntr=0.5,0.3

Type RM Length L Ch R = 1 ,11353   ,114.2,106.2,83.2
BEGIN DESCRIPTION:
structure xs 2; 21.4 ft between structure and xs
END DESCRIPTION:
XS GIS Cut Line= 3
2226781.75931939459612.4760497212226873.36924067459218.155084199
2226694.13243816458807.901958454
#Sta/Elev= 30
       0 2262.82    73.2 2261.99    77.3 2261.38   134.8 2260.38   159.4 2258.31
   415.6 2257.32   458.1  2253.9   482.4 2253.58   494.6 2250.66   505.2 2249.96
   517.7 2248.99   545.6 2249.11     5502249.975   558.7 2253.62   570.5 2254.48
   598.2 2253.69   647.6 2253.68   667.7 2251.75   707.5  2251.9   717.5 2252.44
   737.6 2255.29   747.5 2255.76   757.5 2255.24   764.9    2257   787.5  2257.8
   794.4 2258.82   807.5 2259.51   816.6 2261.84     838 2262.15   852.5 2263.06
#Mann= 7 ,-1,0
       0     .06       0     160     .07       0     170     .06       0
     360      .1       0   505.2    .045       0     550     .06       0
  784.82      .1       0
#XS Ineff= 4 ,-1
  405.63  474.93 2255.21  474.93     498  2250.6     557  571.27  2252.7
  571.27  808.45 2255.21
Permanent Ineff=
       F       F       F       F
Bank Sta=505.2,550
XS Rating Curve= 0 ,0
Exp/Cntr(USF)=0,0
Exp/Cntr=0.5,0.3

Type RM Length L Ch R = 1 ,11247   ,582,564.2,543.4
BEGIN DESCRIPTION:
structure xs 1
END DESCRIPTION:
XS GIS Cut Line= 6
2227023.31295301459602.1203362672227083.02192379459363.739561906
 2227053.2823183459251.7395076922226910.74071235459046.556372116
2226837.56908009458995.5975567942226685.99927042458747.336661637
#Sta/Elev= 30
       0 2266.52      34  2265.2    50.5 2257.82    57.5    2257    71.1 2257.79
    91.7 2256.59   104.1 2258.31   149.9 2260.04   281.5 2258.79   358.1 2256.03
   432.9 2256.14   447.5 2254.85   457.3 2252.43   475.7 2251.16   491.4 2251.85
     506 2250.29   601.9 2252.21   634.4 2250.45   645.92248.193   660.3 2247.54
   668.82248.107   683.3 2251.49   692.6 2249.91   708.2 2251.75   741.7 2249.48
   773.2 2251.72   818.4 2250.41   858.1 2252.14   887.5 2249.32   991.5 2255.32
#Mann= 7 ,-1,0
       0      .1       0  255.74    .025       0  431.63      .1       0
   645.9    .045       0   668.8      .1       0  740.63     .06       0
  850.63      .1       0
#XS Ineff= 2 , 0
                             780            2255
Permanent Ineff=
       F       F
Bank Sta=645.9,668.8
XS Rating Curve= 0 ,0
Exp/Cntr(USF)=0,0
Exp/Cntr=0.3,0.1

Type RM Length L Ch R = 1 ,10683   ,267.5,267.7,267
XS GIS Cut Line= 3
 2227935.8672602459306.2656971832227222.42832575458622.451551517
2226638.96036397458674.165029381
#Sta/Elev= 30
       0 2492.78   110.9  2493.6     199 2486.89   377.3 2481.62   498.2 2473.04
   548.1 2464.48   602.8 2446.74   699.3 2394.88   758.6 2370.65   775.7 2366.58
   808.5 2373.03     821 2372.58   863.9 2361.82   922.8 2339.66   945.5 2324.63
   966.9 2318.69   988.2 2299.33  1014.6 2267.49  1026.6 2243.17  1030.6 2238.99
  1054.7 2237.82  1068.72238.885    1111 2244.97  1139.1 2242.15  1287.7 2247.32
  1428.3    2245  1520.6 2248.25  1540.6 2255.49  1548.7 2256.01    1574 2275.88
#Mann= 7 ,-1,0
       0      .1       0     210     .05       0     320      .1       0
  1030.6    .045       0  1068.7      .1       0 1198.23     .06       0
 1498.23      .1       0
Bank Sta=1030.6,1068.7
XS Rating Curve= 0 ,0
Exp/Cntr(USF)=0,0
Exp/Cntr=0.3,0.1

Type RM Length L Ch R = 1 ,10415   ,537,531.1,524.5
XS GIS Cut Line= 4
2227235.90897364458366.2139840832226986.23619238 458388.24817148
2226933.32177546458363.0508300852226608.53647742458407.976674268
#Sta/Elev= 30
       0 2308.39    15.8  2299.3    43.9 2280.47      68 2258.13    80.1  2247.6
    88.1 2241.68    96.1 2239.23   140.3 2235.75   176.4 2234.92   181.4 2235.82
   188.5 2240.23   200.5 2236.89   212.6 2236.83   224.6 2237.75   236.7 2239.94
   252.9 2240.63   276.4 2239.14   301.7 2240.66     355 2240.53   395.2 2238.76
   463.9 2239.98     480 2238.41   524.4  2240.3   548.7 2240.28   564.8 2243.93
     589 2255.38   597.1 2254.76   601.2 2257.31   613.3    2268   637.1 2281.74
#Mann= 5 ,-1,0
       0      .1       0   140.3    .045       0   181.4      .1       0
  429.25     .06       0  529.25      .1       0
#XS Ineff= 1 ,-1
  254.76   632.4 2249.48
Permanent Ineff=
       F
Bank Sta=140.3,181.4
XS Rating Curve= 0 ,0
Exp/Cntr(USF)=0,0
Exp/Cntr=0.3,0.1

Type RM Length L Ch R = 1 ,9884    ,267.9,272.7,276.8
XS GIS Cut Line= 4
2227306.65150831457891.4898914912227016.57825186457853.597439072
2226895.52576336457900.6796154932226618.89602929457942.267433702
#Sta/Elev= 30
       0 2307.18    26.7    2291    38.8 2282.06      59 2266.56    87.2 2239.39
    97.6 2233.48   115.4 2232.07   139.7 2233.45   167.9 2231.86   216.3  2234.5
   264.7 2230.59   305.8 2231.79   320.12227.466   331.6 2226.13   348.8 2226.18
   353.82227.462   361.6 2230.96   412.8 2233.72   429.9 2233.05   462.2 2228.63
   478.4 2228.16   527.8  2228.6   555.3 2232.03   575.5 2229.34   619.2  2231.9
     624  2235.6   632.1 2245.69   644.2  2256.2   668.6 2273.63   702.2 2300.98
#Mann= 5 ,-1,0
       0      .1       0   320.1    .045       0   353.8      .1       0
  602.42     .06       0  702.16      .1       0
#XS Ineff= 2 ,-1
       0  214.93 2240.63  405.32  563.462261.702
Permanent Ineff=
       F       F
Bank Sta=320.1,353.8
XS Rating Curve= 0 ,0
Exp/Cntr(USF)=0,0
Exp/Cntr=0.3,0.1

Type RM Length L Ch R = 1 ,9611    ,378.8,387.4,397.7
XS GIS Cut Line= 2
2227338.03343575457529.6336102672226502.59369417457677.369068879
#Sta/Elev= 30
       0 2314.57    26.3 2301.52    66.3 2278.66   107.5 2256.97   135.9 2235.63
   148.1 2229.39   200.9 2228.47   232.5 2226.33   395.9 2228.52   412.4 2224.87
   436.1 2223.88   446.5 2224.87   456.8 2228.97   474.1 2228.05   489.3  2231.6
   501.5 2231.52   509.6 2228.52   521.8 2228.12   619.3 2228.25   631.5 2231.01
   647.8 2230.77   655.9 2226.64   659.9 2225.91   692.4 2227.87   732.5 2263.47
   741.2 2270.88   753.7  2284.4   770.9 2300.08   785.9 2312.26   848.4 2358.51
#Mann= 5 ,-1,0
       0      .1       0   412.4    .045       0   446.5      .1       0
   631.5     .06       0   732.5      .1       0
#XS Ineff= 1 ,-1
  493.36  639.53 2232.29
Permanent Ineff=
       T
Bank Sta=412.4,446.5
XS Rating Curve= 0 ,0
Exp/Cntr(USF)=0,0
Exp/Cntr=0.3,0.1

Type RM Length L Ch R = 1 ,9224    ,579.4,563.4,547.5
XS GIS Cut Line= 3
2227330.22322699457293.1288687082226846.19240007457199.313486002
2226457.98429059457349.808472059
#Sta/Elev= 30
       0 2321.98   112.1 2268.84   189.5 2236.41     214 2229.95   234.3 2228.13
   250.6 2221.31   275.6 2222.26   307.7 2220.91   344.3 2222.63   348.4 2222.45
   356.12217.891   360.6 2216.15   376.9 2215.85   390.8 2216.04   397.3 2217.97
   409.5 2223.99   417.7 2225.09   429.9  2222.8   470.6 2221.75   503.8 2222.84
   576.4 2220.49   709.7 2220.23   735.4 2220.77   752.6 2224.63   769.8 2224.45
   774.1 2226.43   782.6 2235.53   842.7 2284.53   872.7 2306.24   909.4 2329.08
#Mann= 6 ,-1,0
       0      .1       0   356.1    .045       0   397.3      .1       0
  523.04     .05       0  733.04     .06       0  843.04      .1       0
#XS Ineff= 2 ,-1
  411.96  621.26 2229.37  725.91  775.75 2233.12
Permanent Ineff=
       F       F
Bank Sta=356.1,397.3
XS Rating Curve= 0 ,0
Exp/Cntr(USF)=0,0
Exp/Cntr=0.3,0.1
